--- DntsRn.prj (project) ---

Proj Title=DntsRn
Current Plan=p01
Default Exp/Contr=0,0
English Units
Geom File=g01
Flow File=f01
Plan File=p01
BEGIN DESCRIPTION:
END DESCRIPTION:
DSS Export Rating Curves= 0
DSS Export Rating Curve Sorted= 0
DSS Export Volume Flow Curves= 0
DXF OffsetX= 0
DXF OffsetY= 0
DXF ScaleX= 0
DXF ScaleY= 0

--- DntsRn.p01 (plan) ---

Plan Title=Floodplain
Program Version=4.00
Geom File=g01
Flow File=f01
K Sum by GR=0
Std Step Tol=0.01
Critical Tol=0.01
Num of Std Step Trials=20
Max Error Tol=0.3
Flow Tol Ratio=0.001
Split Flow NTrial=30
Split Flow Tol=0.02
Split Flow Ratio=0.02
Log Output Level=0
Friction Slope Method=1
Unsteady Friction Slope Method=2
Unsteady Bridges Friction Slope Method=1
Global Log Level=0
CheckData=False
Run HTab=0
Run UNet=0
Run PostProcess=0
UNET Theta=0
UNET Theta Warmup=0
UNET ZTol=0
UNET ZSATol=0
UNET MxIter=0
UNET MaxInSteps=0
UNET DtIC=0
UNET DtMin=0
UNET MaxCRTS=0
UNET WFStab=0
UNET SFStab=0
UNET WFX=0
UNET SFX=0
UNET DSS MLevel=0
UNET DZMax Abort=0
UNET Convert EG Bridges=0
UNET Use Existing IB Tables=0
UNET Froude Limit=0
UNET Froude Power=0
Write IC File=0
Echo Input=False
Echo Output=False
Write Detailed=0

--- DntsRn.f01 (steady flow) ---

Flow Title=NFF Regression Equation
Program Version=4.00
Number of Profiles=1
Profile Names=P100yr
River Rch & RM=DntsRn,Main      ,22812.9
584.1514
River Rch & RM=DntsRn,Main      ,22031.7
627.6647
River Rch & RM=DntsRn,Main      ,21631.7
650.9672
River Rch & RM=DntsRn,Main      ,20431.7
717.7026
River Rch & RM=DntsRn,Main      ,19631.7
776.3647
River Rch & RM=DntsRn,Main      ,17089.9
820.4076
River Rch & RM=DntsRn,Main      ,17089.9
965.1096
River Rch & RM=DntsRn,Main      ,15631.7
1027.066
River Rch & RM=DntsRn,Main      ,15231.7
1375.576
River Rch & RM=DntsRn,Main      ,13631.7
1430.050
River Rch & RM=DntsRn,Main      ,11971.1
1545.186
River Rch & RM=DntsRn,Main      ,6216.3
1672.216
River Rch & RM=DntsRn,Main      ,6031.7
2000.376
River Rch & RM=DntsRn,Main      ,3231.7
2111.543
River Rch & RM=DntsRn,Main      ,31.7
2343.870
River Rch & RM=DntsRn,Main      ,31.7
2345.787
Boundary for River Rch & Prof#=DntsRn,Main      ,1
Up Type=0
Dn Type=3
Dn Slope=0.003406

--- DntsRn.g01 (geometry) ---

Geom Title=USGS 3m DEM
Program Version=4.00

River Reach=DntsRn          ,Main
Reach XY= 30
     1709407.119      390715.256     1709449.037      390558.078
     1709703.694      390416.738     1710119.977      389917.997
     1710304.249      389463.822     1710623.838      389283.299
     1711011.854      388664.322     1711293.718      388574.504
     1711567.358      388121.019     1712109.821      387869.926
     1712854.121      387305.445     1713442.304      386461.302
      1714429.06      385938.516     1714306.216      385750.819
     1714571.941      385192.541     1714617.766       384557.82
     1714871.601      384146.155     1714846.489      383739.116
     1715462.346      382526.903     1715959.715      381814.769
      1717147.19      380942.584      1717817.91      380024.697
     1718905.239      378877.827     1719152.688      378866.048
      1719433.07      378683.643     1720417.805      377819.409
     1721699.589      377463.292     1722194.781      376980.535
      1723388.85      376392.708     1723914.173      375306.387

Type RM Length L Ch R = 1 ,22812.9 ,363.11,381.194,394.075
XS GIS Cut Line= 3
     1709766.545      390978.529     1709448.042      390696.031
     1708970.766      390578.008
#Sta/Elev= 30
       0 1143.11     9.7 1140.59      29 1140.14    38.7  1138.9    48.4 1135.77
    67.7 1132.28    87.1 1132.37   116.1 1128.91   125.8  1126.8   145.1 1127.11
   174.2 1123.64   203.2 1121.87   222.5 1113.08   232.2 1109.93   261.2  1104.9
   280.6 1103.52   309.6 1103.84   338.7    1103   449.1 1094.13   455.2 1093.94
   464.1 1094.33   484.7 1096.62   563.4 1109.66   632.2 1118.57   681.4 1128.48
   691.2 1129.76   710.9 1134.73   760.1 1143.93   838.7 1164.91   917.4 1181.52
#Mann= 3 , 0 , 0
       0      .1       0   449.1    .045       0   464.1      .1       0
Bank Sta=449.1,464.1
XS Rating Curve= 0 ,0
Exp/Cntr=0.3,0.1

Type RM Length L Ch R = 1 ,22431.7 ,414.997,400,396.669
XS GIS Cut Line= 3
     1709887.928      390836.367     1709658.838      390443.541
     1709341.141      390086.493
#Sta/Elev= 30
       0 1127.74    19.4 1127.86    48.4 1125.63    67.7 1126.87   125.8 1126.53
   154.8 1122.11   174.2 1117.19   193.5 1117.43   222.5 1114.06   261.2 1107.78
   299.9 1099.26   367.7 1098.12   447.2  1088.7   454.7  1087.8   462.2 1088.21
   493.8 1094.29     523 1105.05   591.3 1123.89   669.3 1151.86   708.3 1170.57
   737.6 1190.72   766.9 1204.81   786.4 1219.05   805.9 1226.48   835.1 1244.74
   864.4  1256.1   893.7 1272.54   903.4 1273.53   913.2 1277.58   932.7 1289.15
#Mann= 3 , 0 , 0
       0      .1       0   447.2    .045       0   462.2      .1       0
Bank Sta=447.2,462.2
XS Rating Curve= 0 ,0
Exp/Cntr=0.3,0.1

Type RM Length L Ch R = 1 ,22031.7 ,412.563,400,393.965
XS GIS Cut Line= 3
     1710229.084      390451.774     1709888.734      390149.368
     1709539.061      389858.323
#Sta/Elev= 30
       0  1218.3    19.4 1211.39    48.4 1196.15    58.1 1194.72    67.8 1190.37
    87.2 1178.88   106.6 1169.92   135.6  1159.1   164.7 1145.36   184.1 1140.12
   280.9  1096.8   300.3 1093.68   358.4 1092.43   445.6 1083.71   447.8 1083.75
   462.8 1084.74   474.6 1087.53     494 1098.77   542.4 1118.39   581.1 1141.42
   600.5 1147.67   629.5 1164.63   677.9  1188.6   697.3  1200.5   716.6 1208.56
     736 1219.89   755.4 1228.93   784.4 1240.19   813.4 1254.47   910.2 1286.47
#Mann= 3 , 0 , 0
       0      .1       0   447.8    .045       0   462.8      .1       0
Bank Sta=447.8,462.8
XS Rating Curve= 0 ,0
Exp/Cntr=0.3,0.1

Type RM Length L Ch R = 1 ,21631.7 ,460.651,466.364,464.682
XS GIS Cut Line= 3
     1710588.784      389934.675     1710144.889      389853.974
     1709712.022      389654.307
#Sta/Elev= 30
       0 1166.76    39.2  1154.5   107.9 1138.28   117.7 1134.53   147.1 1118.46
   156.9 1111.66   166.7  1107.7   225.6 1098.72   411.9 1087.09   443.7 1083.19
   451.2 1082.96   458.7 1084.59   480.4 1095.95   509.5 1115.21   519.3 1118.48
   538.7  1130.1   548.5 1132.87   567.9 1144.18   587.4 1151.47   606.8 1161.92
   616.6 1164.58     636 1175.39   704.1 1202.85   723.6 1208.46   772.2 1227.14
   811.1 1234.97   840.3 1236.23   879.2  1232.4   908.4  1233.4   927.9 1230.12
#Mann= 3 , 0 , 0
       0      .1       0   443.7    .045       0   458.7      .1       0
Bank Sta=443.7,458.7
XS Rating Curve= 0 ,0
Exp/Cntr=0.3,0.1

Type RM Length L Ch R = 1 ,21165.4 ,325.593,333.636,344.193
XS GIS Cut Line= 3
     1710641.438      389812.322     1710373.085      389469.102
     1709924.411      389225.378
#Sta/Elev= 30
       0 1176.48    67.8 1153.11    96.8 1141.54   106.5 1137.24   125.9 1124.42
   145.2 1113.79   154.9 1110.06   164.6 1109.01   174.3 1105.89   193.6 1096.56
   222.7 1084.61   232.4 1082.31   271.1 1079.51   396.9 1078.76   465.1 1076.78
   466.5 1076.95     475 1077.99   481.5 1080.84   484.8 1082.28   504.4 1096.69
   573.1 1102.68   612.4 1102.61   651.7 1106.79   671.3  1111.7   749.9 1122.85
   769.5 1124.53   808.8 1134.38   838.3 1138.56   897.2 1153.27   946.3 1162.45
#Mann= 3 , 0 , 0
       0      .1       0   466.5    .045       0   481.5      .1       0
Bank Sta=466.5,481.5
XS Rating Curve= 0 ,0
Exp/Cntr=0.3,0.1

Type RM Length L Ch R = 1 ,20831.7 ,403.902,400,395.082
XS GIS Cut Line= 3
     1710943.621      389593.734     1710625.485      389280.743
     1710306.227      388941.246
#Sta/Elev= 30
       0 1130.73     9.7  1129.6    38.8  1132.5    87.3 1132.01   106.7 1129.31
   184.3 1126.05     194 1123.43   232.8 1101.62     262 1096.29   281.4 1083.26
   291.1 1079.52   378.4  1076.8   438.8 1071.11   446.3 1070.99   453.8 1072.16
   465.7  1078.1   475.4 1087.37   504.5 1104.55   533.7 1113.97   601.6  1145.4
   630.8 1155.67   659.9 1171.17   679.3 1176.46   708.4 1190.23   737.6 1200.82
   805.5 1231.37   824.9 1244.32   873.5 1261.78   892.9  1266.5   912.3 1275.09
#Mann= 3 , 0 , 0
       0      .1       0   438.8    .045       0   453.8      .1       0
Bank Sta=438.8,453.8
XS Rating Curve= 0 ,0
Exp/Cntr=0.3,0.1

Type RM Length L Ch R = 1 ,20431.7 ,361.468,365.345,369.317
XS GIS Cut Line= 3
     1711220.239      389207.262     1710846.319       388947.72
     1710471.467      388689.876
#Sta/Elev= 30
       0 1167.27    29.1 1163.17   106.5 1143.31     155 1125.03   174.3 1120.34
     184 1116.01   203.4 1103.29   232.4 1081.52   242.1 1079.08   445.5 1066.48
   447.7 1066.52   462.7  1068.4   474.5 1074.75   493.9 1092.31   513.2 1101.14
   532.6 1113.44   542.3 1117.04   561.6 1130.78     581 1137.75   600.4 1151.63
   639.1 1171.45   648.8 1173.03   687.5 1191.72   726.2 1207.29   755.3 1223.63
   803.7 1242.26     823 1251.98   861.7 1265.17   890.8 1269.03   910.1 1268.52
#Mann= 3 , 0 , 0
       0      .1       0   447.7    .045       0   462.7      .1       0
Bank Sta=447.7,462.7
XS Rating Curve= 0 ,0
Exp/Cntr=0.3,0.1

Type RM Length L Ch R = 1 ,20066.4 ,434.961,434.655,429.956
XS GIS Cut Line= 3
     1711406.143       389006.58     1710985.165      388591.142
     1710600.192      388441.584
#Sta/Elev= 30
       0 1121.36     126 1114.52   145.4 1110.09   174.5 1108.46   193.9 1102.25
   213.3 1099.78   252.1  1090.8   281.2 1073.52   300.6 1070.75   475.1    1069
   494.5 1067.33   509.2 1064.32   513.9 1063.44   524.2 1064.01     543  1075.2
   572.1 1087.84   591.4 1092.92   611.1 1100.93   660.3 1116.06   679.9 1124.68
   689.8 1125.84   709.4 1131.41   748.8 1138.32   807.8 1142.84     857 1144.34
   886.5  1148.9   906.1 1150.29   945.5 1152.26   955.3 1151.34  1004.5 1156.58
#Mann= 3 , 0 , 0
       0      .1       0   509.2    .045       0   524.2      .1       0
Bank Sta=509.2,524.2
XS Rating Curve= 0 ,0
Exp/Cntr=0.3,0.1

Type RM Length L Ch R = 1 ,19631.7 ,396.374,400,410.753
XS GIS Cut Line= 3
      1711721.28      388741.943     1711378.777      388443.075
     1711001.941      388138.023
#Sta/Elev= 30
       0 1263.74      29 1251.41      58 1241.89      87 1227.76   135.4  1209.6
   154.7 1200.79   174.1 1195.52   232.1 1171.25   270.8 1151.32   290.1 1144.39
   328.8 1121.42   348.2 1115.05   406.2 1076.39   447.1 1060.62   454.6 1059.16
   462.1 1059.36   522.4 1067.23   561.2 1069.14   638.8 1068.41     697 1070.94
   735.8  1075.3   774.6 1093.17   793.9 1106.15   813.3 1116.54   852.1 1132.45
   871.5 1142.74   881.2    1146   890.9 1147.12     920 1160.99   939.4 1167.62
#Mann= 3 , 0 , 0
       0      .1       0   447.1    .045       0   462.1      .1       0
Bank Sta=447.1,462.1
XS Rating Curve= 0 ,0
Exp/Cntr=0.3,0.1

Type RM Length L Ch R = 1 ,19231.7 ,389.803,400,399.364
XS GIS Cut Line= 3
     1711880.265      388498.676       1711571.4       388118.78
     1711333.551      387738.139
#Sta/Elev= 30
       0  1218.9    19.6 1208.53    39.2 1201.85    68.5 1185.29    88.1 1179.25
   117.5 1165.36   137.1 1159.92   166.5 1143.74   186.1 1135.51   215.4  1116.3
     235 1108.14   254.6 1095.05   264.4 1091.47     284 1088.93   323.1  1070.7
   362.3 1061.26   450.4 1062.61   482.1  1057.3   489.6 1055.12   497.1 1055.69
   577.4 1069.11   655.5 1089.54   723.8 1102.98   753.1 1111.06   792.1 1128.55
   811.6 1134.34   840.9 1147.07   850.6 1148.31   879.9 1162.03   938.5 1181.11
#Mann= 3 , 0 , 0
       0      .1       0   482.1    .045       0   497.1      .1       0
Bank Sta=482.1,497.1
XS Rating Curve= 0 ,0
Exp/Cntr=0.3,0.1

Type RM Length L Ch R = 1 ,18831.7 ,404.847,400,392.965
XS GIS Cut Line= 3
     1712089.454      388388.411     1711907.982      387966.402
     1711716.755      387546.718
#Sta/Elev= 30
       0  1196.2    48.9 1184.97    68.4 1175.54    78.2 1174.24   107.5 1160.63
   136.8 1149.94   156.4 1138.07   166.2 1136.26   195.5 1116.96     215 1108.66
   234.6 1096.72   244.3 1093.65   263.9 1090.98   293.2 1075.57     303 1067.87
   312.8  1062.6   451.9 1051.05   459.4 1050.99   466.9 1051.64   498.6  1060.4
   508.4 1060.91   577.1 1077.45   685.1 1098.32   704.7 1104.26   724.3  1107.5
     793 1130.11   851.9  1144.1   871.5 1151.99   891.1 1157.45   920.6 1172.14
#Mann= 3 , 0 , 0
       0      .1       0   451.9    .045       0   466.9      .1       0
Bank Sta=451.9,466.9
XS Rating Curve= 0 ,0
Exp/Cntr=0.3,0.1

Type RM Length L Ch R = 1 ,18431.7 ,400.895,400,401.702
XS GIS Cut Line= 3
     1712510.277      388132.057     1712239.979      387764.518
     1711928.583      387428.554
#Sta/Elev= 30
       0 1179.76    19.4  1173.9    58.2 1153.03    77.7 1146.61   106.8 1127.69
   116.5 1124.72   135.9 1108.48   145.6 1102.32   174.7 1094.09   203.8 1076.74
   252.4 1063.26   291.2 1058.01     330  1056.6   388.3 1058.05   407.7 1056.94
   448.7 1049.91   456.2 1049.37   463.7 1049.84     505 1058.59   543.9 1069.16
   573.2 1072.36   660.9 1092.22   670.7 1092.73   699.9 1100.91   719.4 1104.01
   836.3 1130.63   846.1 1133.33   875.3 1147.45   885.1 1149.01   914.3 1163.85
#Mann= 3 , 0 , 0
       0      .1       0   448.7    .045       0   463.7      .1       0
Bank Sta=448.7,463.7
XS Rating Curve= 0 ,0
Exp/Cntr=0.3,0.1

Type RM Length L Ch R = 1 ,18031.7 ,406.144,400,397.132
XS GIS Cut Line= 3
     1712820.351      387869.437     1712539.335       387511.59
     1712258.318      387153.742
#Sta/Elev= 30
       0 1155.83      29 1141.35    48.4 1135.38    77.4 1115.41   106.5 1099.76
   145.2 1090.67   174.3 1076.69   193.6 1071.64   222.7 1058.56   232.3 1056.07
   261.4 1050.08   447.5 1044.18     455 1044.08   462.5 1045.93   493.7 1055.65
   522.8 1069.08   542.1 1073.24   571.2 1084.17   590.5 1087.44   619.6 1097.52
   687.3 1114.13   735.7 1132.36   774.5 1153.33   784.1 1155.52   793.8 1160.41
   822.9 1177.97   842.2 1185.09   871.3 1203.61   890.6 1210.38     910 1223.39
#Mann= 3 , 0 , 0
       0      .1       0   447.5    .045       0   462.5      .1       0
Bank Sta=447.5,462.5
XS Rating Curve= 0 ,0
Exp/Cntr=0.3,0.1

Type RM Length L Ch R = 1 ,17631.7 ,545.621,541.866,534.835
XS GIS Cut Line= 3
     1713229.543      387557.039     1712866.936      387288.163
     1712529.919      386953.015
#Sta/Elev= 30
       0 1101.89    19.6 1102.58    68.7  1113.3    78.5 1113.94   137.4 1098.72
   147.2  1094.7   186.5  1071.5   215.9 1066.39   235.5 1056.43     265 1047.89
     314 1046.92   382.7 1047.99   443.9 1042.77   451.4 1042.38   458.9 1042.95
   519.3 1054.94   548.4 1064.03   567.8  1068.2   596.9 1078.09   616.3 1082.03
   693.9 1108.47   713.3  1118.9   732.7 1126.11   761.8 1142.67   790.9 1152.66
   810.3 1161.32   839.4 1170.73   878.2 1190.19   907.3 1208.67   926.7 1227.11
#Mann= 3 , 0 , 0
       0      .1       0   443.9    .045       0   458.9      .1       0
Bank Sta=443.9,458.9
XS Rating Curve= 0 ,0
Exp/Cntr=0.3,0.1

Type RM Length L Ch R = 1 ,17089.9 ,328.597,340.631,349.532
XS GIS Cut Line= 3
     1713409.462      387314.976     1713281.689      386928.675
     1712746.797      386664.537
#Sta/Elev= 30
       0 1058.71    29.1 1058.21   106.6 1061.02     155 1060.19   222.8 1054.09
   251.9 1053.48   271.3  1051.2   377.8 1045.15   426.4 1043.88   520.1 1038.43
   524.2 1038.27   535.1  1038.4   631.8 1043.28   651.4 1046.77   661.2 1050.13
   680.7 1064.85   710.1 1083.67   739.4  1094.8   768.7  1104.4   778.5  1106.5
   798.1 1108.09     847 1119.59   866.5 1121.83   876.3  1124.4   895.9 1126.32
   915.4 1133.03   944.8 1138.02   964.3 1139.45   983.9 1144.71  1003.4 1148.29
#Mann= 3 , 0 , 0
       0      .1       0   520.1    .045       0   535.1      .1       0
Bank Sta=520.1,535.1
XS Rating Curve= 0 ,0
Exp/Cntr=0.3,0.1

Type RM Length L Ch R = 1 ,16749.2 ,309.785,317.503,321.423
XS GIS Cut Line= 3
     1713676.236      386904.362     1713382.395      386673.037
     1713041.544      386316.694
#Sta/Elev= 30
       0 1100.14    28.8 1095.22    76.7 1080.17    86.3  1078.9   124.7 1065.01
   134.2 1063.06   143.8 1059.57     163 1050.61   172.6 1048.25   239.7 1043.82
     403 1043.92     461 1040.66   475.3 1038.08     490 1037.21   490.3 1037.24
   567.3 1045.96     606 1053.85   644.7 1068.67   654.4 1071.59   673.7 1075.25
   702.7 1085.86   712.4 1086.77     722 1089.61   760.7 1106.68   770.4  1109.3
   789.7 1111.94   809.1 1116.19   828.4 1117.02   847.7 1119.64   867.1 1125.67
#Mann= 3 , 0 , 0
       0      .1       0   475.3    .045       0   490.3      .1       0
Bank Sta=475.3,490.3
XS Rating Curve= 0 ,0
Exp/Cntr=0.3,0.1

Type RM Length L Ch R = 1 ,16431.7 ,406.05,400,399.927
XS GIS Cut Line= 3
     1713758.153      386829.162     1713543.856      386406.739
     1713288.458      386031.717
#Sta/Elev= 30
       0 1093.67    48.3 1080.17    67.7 1076.55    96.7 1067.33     116 1063.58
   164.3  1048.7     174  1047.5     203 1046.32   251.3 1041.23   367.3 1040.57
   466.2 1036.89   473.7 1036.61   481.2 1037.45   512.3 1046.97   531.6 1056.08
   550.9 1062.68   589.5 1080.59   608.8 1087.17   628.1 1097.38   657.1 1107.44
   686.1 1122.77   705.4 1129.45   724.7 1141.07   753.6 1153.77   782.6 1169.13
   830.9 1189.84   859.8 1206.84   898.4 1220.98   917.7 1223.66   927.4 1227.22
#Mann= 3 , 0 , 0
       0      .1       0   466.2    .045       0   481.2      .1       0
Bank Sta=466.2,481.2
XS Rating Curve= 0 ,0
Exp/Cntr=0.3,0.1

Type RM Length L Ch R = 1 ,16031.7 ,387.084,400,392.408
XS GIS Cut Line= 3
     1714162.246      386570.833     1713867.866      386219.825
      1713618.27      385838.891
#Sta/Elev= 30
       0 1125.26      39 1108.94    97.5 1088.28   136.5 1072.76   185.2 1059.07
   204.7 1055.91   243.7 1053.01   263.2 1049.16   292.4 1039.81   370.4 1037.49
   450.6 1031.29   458.1  1031.2   465.6 1032.12   487.2 1042.71   506.6  1048.8
   535.6 1062.97   564.7 1069.15   593.8 1082.51   632.5  1092.9   690.7 1104.24
   729.4 1117.83   739.1 1119.01   768.2  1130.4   787.6 1134.49   826.3 1147.76
     836 1148.59   845.7 1151.46   884.5 1164.44   903.8 1173.76   913.5 1176.38
#Mann= 3 , 0 , 0
       0      .1       0   450.6    .045       0   465.6      .1       0
Bank Sta=450.6,465.6
XS Rating Curve= 0 ,0
Exp/Cntr=0.3,0.1

Type RM Length L Ch R = 1 ,15631.7 ,439.4,400,383.253
XS GIS Cut Line= 3
     1714282.925      386497.395      1714223.07      386056.356
     1713840.423      385690.217
#Sta/Elev= 30
       0 1134.42    38.7 1116.27   116.1 1094.52   164.5  1082.7   193.5 1073.22
   212.9 1068.78   232.2 1061.05   241.9 1059.45   261.2  1052.3   290.3  1049.1
   309.6 1042.84   338.6 1038.38   437.6 1029.75   445.1  1029.6   452.6 1029.79
   484.3 1031.66   523.5 1036.35   582.4 1051.27     602 1054.02   631.4  1062.3
   670.7 1070.67   690.3 1073.38   749.1 1095.48   778.5    1103     808 1113.31
   837.4 1119.46   896.2 1136.52   925.6 1149.31   945.3 1154.43   974.7 1167.78
#Mann= 3 , 0 , 0
       0      .1       0   437.6    .045       0   452.6      .1       0
Bank Sta=437.6,452.6
XS Rating Curve= 0 ,0
Exp/Cntr=0.3,0.1

Type RM Length L Ch R = 1 ,15231.7 ,390.571,400,394.956
XS GIS Cut Line= 3
     1714842.941      385786.305     1714334.371      385828.131
     1713885.807      385631.755
#Sta/Elev= 30
       0 1062.37    68.7 1061.62    98.1 1060.06   137.4 1054.04   166.8 1050.86
   225.7 1041.29   245.3 1037.18     265  1034.8   294.4 1033.89     471 1034.03
   502.8 1029.68   510.3 1028.88   517.8 1028.93   529.9 1029.09     569 1032.12
   598.4 1037.56   627.8 1048.73   647.4 1060.87   676.8 1072.21   696.4 1077.65
   735.5    1092   745.3 1096.27   755.1 1098.84   784.5 1111.45   813.9 1118.95
   833.5 1125.64   853.1 1133.37   892.2  1142.8     951 1161.82    1000  1174.9
#Mann= 3 , 0 , 0
       0      .1       0   502.8    .045       0   517.8      .1       0
#XS Ineff= 2 , 0
          372.75 1034.46
Permanent Ineff=
       F       F
Bank Sta=502.8,517.8
XS Rating Curve= 0 ,0
Exp/Cntr=0.3,0.1

Type RM Length L Ch R = 1 ,14831.7 ,401.707,400,398.097
XS GIS Cut Line= 3
     1714897.091      385615.048     1714461.869      385481.682
     1714028.993      385341.016
#Sta/Elev= 30
       0 1084.94    67.8 1077.25   164.6  1059.9     184 1053.99   222.8  1046.4
   242.1 1036.05   251.8 1032.35   261.5 1030.89   387.4 1029.81   426.1 1027.64
   447.7 1024.59   455.2 1024.21   462.7 1026.68   474.6 1033.64   513.3 1035.19
     523 1036.99     552 1050.81   581.1 1072.52   590.8 1083.54   600.5 1090.79
   648.9 1096.23   677.9 1108.01     707 1121.41   726.4 1133.22   745.7 1141.34
   774.8 1156.58   794.1 1168.43   803.8 1170.83   852.2 1194.19   910.4 1218.83
#Mann= 3 , 0 , 0
       0      .1       0   447.7    .045       0   462.7      .1       0
#XS Ineff= 2 , 0
          310.97 1031.14
Permanent Ineff=
       F       F
Bank Sta=447.7,462.7
XS Rating Curve= 0 ,0
Exp/Cntr=0.3,0.1

Type RM Length L Ch R = 1 ,14431.7 ,405.66,400,391.013
XS GIS Cut Line= 3
      1715028.54      385209.337     1714582.038      385105.785
     1714140.229       384999.52
#Sta/Elev= 30
       0 1150.78    48.8 1134.93      78 1120.42   146.3 1100.89   165.8 1090.83
   175.5 1089.12   185.3 1083.82   204.8 1077.43   224.3 1068.48   273.1    1055
   312.1 1034.26   321.8 1032.25   429.1 1027.28   450.9 1021.54   458.4 1019.53
   465.9 1020.71   477.7 1026.79   506.7 1033.73   535.7 1036.19     584  1035.6
     613 1051.13   632.4 1065.69     642  1068.7   661.4    1083   680.7 1090.18
   767.7 1109.78   787.1 1117.19   854.8  1136.1   883.8 1139.66   912.8 1140.72
#Mann= 3 , 0 , 0
       0      .1       0   450.9    .045       0   465.9      .1       0
Bank Sta=450.9,465.9
XS Rating Curve= 0 ,0
Exp/Cntr=0.3,0.1

Type RM Length L Ch R = 1 ,14031.7 ,389.405,400,413.738
XS GIS Cut Line= 3
     1715106.548       384703.17     1714641.225      384719.254
     1714181.621      384793.461
#Sta/Elev= 30
       0 1176.74     9.7  1173.5    29.1 1163.38    58.2 1154.07      97 1146.06
   155.2 1123.42     194 1111.97   271.6 1079.69   281.3 1076.88   300.7 1066.24
   329.8 1053.11   339.5 1050.17   358.9 1039.04   368.6 1035.16   397.7 1032.44
   426.8 1024.77   458.1 1019.48   465.6 1019.17   473.1 1020.49     485 1025.74
   504.4 1028.97   649.9 1035.14   708.1 1034.72   717.8 1037.72   737.2 1048.25
   756.6 1056.43   795.4 1067.94   814.8 1069.59   853.6 1078.59   931.2 1082.68
#Mann= 3 , 0 , 0
       0      .1       0   458.1    .045       0   473.1      .1       0
Bank Sta=458.1,473.1
XS Rating Curve= 0 ,0
Exp/Cntr=0.3,0.1

Type RM Length L Ch R = 1 ,13631.7 ,412.326,400,390.982
XS GIS Cut Line= 3
     1715153.212      384565.204     1714743.304      384367.718
     1714333.396      384170.232
#Sta/Elev= 30
       0 1203.01    38.7 1189.42    96.8 1161.55   116.2 1149.21   154.9 1130.18
   203.3 1114.89   271.1 1088.49   290.4 1074.81   309.8 1064.87   329.1 1052.29
   348.5 1043.01   377.6 1037.89   396.9 1029.76   447.5 1018.36   462.5    1017
   464.7 1016.98   503.4 1021.85   551.8 1031.91   571.2 1030.93   590.5 1024.07
   609.9 1021.62   716.4 1030.17   745.4 1039.36   764.8 1051.53   774.5 1054.95
   793.8 1065.93   822.9 1078.05   842.2 1083.65   861.6 1091.65     910 1105.97
#Mann= 3 , 0 , 0
       0      .1       0   447.5    .045       0   462.5      .1       0
#XS Ineff= 2 , 0
                          561.56         1031.58
Permanent Ineff=
       F       F
Bank Sta=447.5,462.5
XS Rating Curve= 0 ,0
Exp/Cntr=0.3,0.1

Type RM Length L Ch R = 1 ,13231.7 ,389.582,400,410.085
XS GIS Cut Line= 3
      1715330.23      383962.005      1714882.53      384007.277
     1714399.596      383985.436
#Sta/Elev= 30
       0 1087.46   117.4  1065.1   176.1 1047.04   195.6 1039.74   244.6 1040.31
   264.1 1034.57   293.5 1030.17   371.7 1034.31   391.3 1034.02   420.6 1024.51
   442.5 1014.91     450 1012.88   457.5 1013.39   488.7 1018.91   527.3 1029.81
     537 1030.48   546.7 1030.01   575.7  1024.7   604.7 1017.23   614.3 1016.62
   633.7  1018.5   672.4 1031.18     682 1035.95   701.4 1042.47   720.7 1051.67
   730.4 1053.53   778.7 1072.39   817.4 1082.53   875.4 1101.39   933.4 1124.68
#Mann= 3 , 0 , 0
       0      .1       0   442.5    .045       0   457.5      .1       0
#XS Ineff= 2 , 0
                          539.42         1030.58
Permanent Ineff=
       F       F
Bank Sta=442.5,457.5
XS Rating Curve= 0 ,0
Exp/Cntr=0.3,0.1

Type RM Length L Ch R = 1 ,12831.7 ,403.247,406.963,407.703
XS GIS Cut Line= 3
     1715334.496      383791.538     1714903.507      383631.419
     1714546.859      383442.472
#Sta/Elev= 30
       0 1046.64    97.8 1042.84   107.6 1041.43   146.7 1027.53   156.5 1026.54
     225 1033.82   342.4 1032.37   401.1  1029.6   420.6 1026.07   452.3 1012.67
   459.8 1012.14   467.3 1013.05     479 1017.12   517.4  1038.2   546.3 1050.93
   555.9 1053.01   584.7    1067   642.4 1091.22   671.2 1107.42   690.4 1120.61
     700  1124.1   719.2 1136.39   738.5  1145.1   757.7 1158.39   767.3 1161.35
   786.5 1172.43   805.7 1180.34   824.9 1191.68   834.5 1194.42   863.4 1209.95
#Mann= 3 , 0 , 0
       0      .1       0   452.3    .045       0   467.3      .1       0
Bank Sta=452.3,467.3
XS Rating Curve= 0 ,0
Exp/Cntr=0.3,0.1

Type RM Length L Ch R = 1 ,12424.8 ,453.202,453.679,454.157
XS GIS Cut Line= 3
     1715484.963      383496.217     1715042.616      383243.061
      1714610.56      383331.688
#Sta/Elev= 30
       0 1051.97    39.2 1041.55    78.4 1038.56    88.2 1034.41      98 1025.72
   107.8 1021.57   117.6 1023.59   137.2 1032.29     147 1032.93   186.2  1029.8
   235.2 1021.65   264.6 1019.29   362.6 1016.66   392.1 1019.42   447.6 1012.28
   460.7 1011.84   462.6 1012.33   470.5 1014.39   490.1 1027.32   519.5 1040.04
   568.5 1054.37   597.9 1063.93   617.5 1072.95   627.3 1074.09   656.7 1084.22
   676.3 1093.16   823.3 1148.82   862.5 1160.43   931.1 1173.96   950.7 1180.37
#Mann= 3 , 0 , 0
       0      .1       0   447.6    .045       0   462.6      .1       0
#XS Ineff= 2 , 0
          394.15 1019.74
Permanent Ineff=
       F       F
Bank Sta=447.6,462.6
XS Rating Curve= 0 ,0
Exp/Cntr=0.3,0.1

Type RM Length L Ch R = 1 ,11971.1 ,340.606,339.358,338.11
XS GIS Cut Line= 3
     1715686.215      383102.707     1715255.874       382844.24
     1714807.201      382852.549
#Sta/Elev= 30
       0  1037.2     9.7  1037.8    19.3 1036.93    38.6 1032.34    57.9 1026.07
    77.2 1017.38    86.9  1015.2   125.5 1018.66   289.6 1018.09   347.5 1010.72
   357.2 1011.27   376.5 1020.05   386.1 1023.25   405.5 1024.28   424.8 1021.88
   434.4 1018.98   451.5    1011   463.4  1008.9   466.5 1009.57     473 1010.97
   482.7 1016.01   521.5 1027.82     541 1031.64     580 1036.23   658.1 1038.89
   706.9 1043.05   736.1 1039.14   755.6 1038.39   823.9 1043.89   950.7  1050.6
#Mann= 3 , 0 , 0
       0      .1       0   451.5    .045       0   466.5      .1       0
#XS Ineff= 2 , 0
          407.44 1024.24
Permanent Ineff=
       F       F
Bank Sta=451.5,466.5
XS Rating Curve= 0 ,0
Exp/Cntr=0.3,0.1

Type RM Length L Ch R = 1 ,11631.7 ,442.904,446.672,450.44
XS GIS Cut Line= 3
     1715845.715      382775.297     1715443.393      382562.784
     1715041.071      382350.271
#Sta/Elev= 30
       0 1026.23    19.4 1016.71      29 1014.74    96.8  1017.5   154.9  1017.5
   319.5 1010.77   329.1 1010.78   377.6  1022.7   396.9 1023.34     426 1016.99
   447.5 1008.83     455 1008.01   462.5 1009.48   474.4 1017.42     484  1027.1
   493.7 1030.75   513.1  1043.4   542.1 1048.67   561.5 1054.83   580.9 1064.29
   600.2  1071.4   638.9 1091.86   648.6 1100.18   677.7 1118.49     697 1127.92
   764.8  1152.1   803.5 1161.01   861.6 1178.34   871.3 1179.69     910 1192.15
#Mann= 3 , 0 , 0
       0      .1       0   447.5    .045       0   462.5      .1       0
#XS Ineff= 2 , 0
          395.93 1024.21
Permanent Ineff=
       F       F
Bank Sta=447.5,462.5
XS Rating Curve= 0 ,0
Exp/Cntr=0.3,0.1

Type RM Length L Ch R = 1 ,11185.1 ,363.056,363.77,364.485
XS GIS Cut Line= 3
     1716029.227      382501.414     1715710.087      382207.234
     1715372.197      381949.662
#Sta/Elev= 30
       0 1021.54     9.6 1016.47    19.3 1013.86    57.9 1017.65     164 1016.95
   279.7 1014.61   356.9 1009.85   366.5 1010.89   405.1 1020.78   414.8 1020.14
     434 1014.42   453.9  1005.6     463 1004.97   468.9 1006.15   482.3 1012.58
   501.6 1030.15   520.9 1041.38   530.6 1048.91   578.9 1072.66   588.5 1073.56
   617.5 1070.62   646.5 1059.28   656.1 1057.64   723.7 1054.34     743  1055.7
   762.3  1060.8   791.3 1076.81   810.6 1081.37   839.6 1093.95   858.9 1098.58
#Mann= 3 , 0 , 0
       0      .1       0   453.9    .045       0   468.9      .1       0
#XS Ineff= 2 , 0
          404.78 1020.92
Permanent Ineff=
       F       F
Bank Sta=453.9,468.9
XS Rating Curve= 0 ,0
Exp/Cntr=0.3,0.1

Type RM Length L Ch R = 1 ,10821.3 ,383.711,389.558,395.404
XS GIS Cut Line= 3
     1716248.562      382180.629     1715870.724      381872.113
     1715740.553      381484.371
#Sta/Elev= 30
       0 1025.51      39  1013.9   107.3  1017.4   273.2 1017.48   312.2  1014.7
   351.2 1006.44     361 1007.08     400 1018.41   409.7 1018.03     439 1006.66
   447.5  1005.2   458.5 1004.97   462.5 1005.08     478 1007.89     517 1043.59
   526.7 1049.78   575.4 1068.86   604.7 1073.93   633.9 1074.68   653.3 1080.82
   682.6 1085.71     702 1093.65   731.3 1101.25   760.5 1105.31   789.7 1123.28
   799.4 1125.19   818.9 1133.51   838.4 1139.07   867.6 1155.12   896.8 1162.95
#Mann= 3 , 0 , 0
       0      .1       0   447.5    .045       0   462.5      .1       0
#XS Ineff= 2 , 0
          401.24 1018.71
Permanent Ineff=
       F       F
Bank Sta=447.5,462.5
XS Rating Curve= 0 ,0
Exp/Cntr=0.3,0.1

Type RM Length L Ch R = 1 ,10431.7 ,399.889,400,400.111
XS GIS Cut Line= 3
     1716459.483      382014.345     1716192.674      381645.784
     1715925.864      381277.223
#Sta/Elev= 30
       0 1024.86     9.7 1023.26      29 1014.46    38.7 1012.47   203.3 1011.93
   348.5 1004.29   358.2 1005.91   377.6 1014.87   396.9 1017.87   416.3 1014.57
   435.6 1006.26   447.5 1005.12   462.5 1005.97   464.7 1006.26   474.4 1013.21
     484 1022.35   493.7 1027.96   532.4 1068.14   551.8 1074.76   638.9 1088.59
   648.6 1089.55     668 1088.11   687.3 1089.99   735.7 1086.17   764.8 1079.89
   793.8 1077.49   822.9 1072.19   842.2 1072.72     881 1081.51     910 1093.85
#Mann= 3 , 0 , 0
       0      .1       0   447.5    .045       0   462.5      .1       0
#XS Ineff= 2 , 0
           397.7 1018.42
Permanent Ineff=
       F       F
Bank Sta=447.5,462.5
XS Rating Curve= 0 ,0
Exp/Cntr=0.3,0.1

Type RM Length L Ch R = 1 ,10031.7 ,400.681,400,399.319
XS GIS Cut Line= 3
     1716785.733      381787.705     1716520.762      381417.819
     1716255.791      381047.933
#Sta/Elev= 30
       0 1022.27      29 1020.26    48.4 1009.67    58.1 1008.37   106.5 1012.08
   183.9  1013.9   280.7 1010.81   348.5 1004.88   358.2 1005.56   387.2 1015.35
   406.6 1016.22   447.5 1005.33     455 1004.84   462.5 1005.71   474.4 1010.74
   493.7 1025.38   503.4 1027.25   522.8 1055.48   532.4 1066.23   542.1 1072.84
   571.2 1083.82   590.5 1094.03   629.3  1102.6   677.7 1125.89     697 1129.36
   745.4 1146.61   784.1 1164.97   793.8 1165.83   822.9 1178.09     910 1192.45
#Mann= 3 , 0 , 0
       0      .1       0   447.5    .045       0   462.5      .1       0
#XS Ineff= 2 , 0
          400.35 1017.11
Permanent Ineff=
       F       F
Bank Sta=447.5,462.5
XS Rating Curve= 0 ,0
Exp/Cntr=0.3,0.1

Type RM Length L Ch R = 1 ,9631.7  ,403.472,400,396.73
XS GIS Cut Line= 3
     1717125.502      381551.729     1716849.462       381190.03
     1716573.421      380828.331
#Sta/Elev= 30
       0 1027.62     9.7 1020.89    48.4 1019.19    77.4  1007.6   106.5 1012.35
   154.9 1012.86   348.5 1004.82   396.9 1015.38   416.3 1012.48   447.5 1001.09
     455   999.9   462.5 1000.19   474.4 1003.32   503.4 1020.32   522.8 1028.93
   542.1 1041.95   561.5 1049.18   590.5 1066.97   619.6 1079.87   638.9  1092.2
   687.3  1114.1   716.4 1124.29   735.7 1134.45   764.8  1144.1   793.8 1158.81
   813.2 1165.44   832.6  1176.8   861.6 1187.51   900.3 1207.56     910 1209.12
#Mann= 3 , 0 , 0
       0      .1       0   447.5    .045       0   462.5      .1       0
#XS Ineff= 2 , 0
          398.58 1016.32
Permanent Ineff=
       F       F
Bank Sta=447.5,462.5
XS Rating Curve= 0 ,0
Exp/Cntr=0.3,0.1

Type RM Length L Ch R = 1 ,9231.7  ,404.323,400,395.475
XS GIS Cut Line= 3
     1717484.201      381248.527     1717155.858      380933.547
     1716830.336      380615.616
#Sta/Elev= 30
       0 1018.54    38.7 1016.77    67.8 1004.99    87.1 1003.77     242 1003.92
   300.1 1005.83   338.8 1001.96   358.2 1011.66   367.9 1014.56   387.2 1015.71
   396.9 1014.64   447.5 1000.43     455  999.19   462.5 1000.84   464.7 1001.33
     484 1020.09   493.7 1026.39   503.4 1029.81   532.4 1053.43   551.8 1061.54
   571.2 1077.05   600.2 1095.52   648.6 1122.18     668 1124.06   735.8 1120.91
   764.8 1117.39   784.2 1118.72   813.2 1115.49   890.7 1115.33     910 1111.49
#Mann= 3 , 0 , 0
       0      .1       0   447.5    .045       0   462.5      .1       0
#XS Ineff= 2 , 0
           385.3 1015.79
Permanent Ineff=
       F       F
Bank Sta=447.5,462.5
XS Rating Curve= 0 ,0
Exp/Cntr=0.3,0.1

Type RM Length L Ch R = 1 ,8831.7  ,398.842,400,401.044
XS GIS Cut Line= 3
     1717761.403      380849.947     1717378.995      380603.392
     1716996.587      380356.837
#Sta/Elev= 30
       0 1078.91    38.7 1058.75    48.4 1056.18    77.4 1043.45   106.5 1028.76
   116.2 1027.32   154.9 1016.62   183.9 1005.12   193.6 1003.78   261.4 1001.46
   329.1 1000.68   367.9 1010.12   396.9 1013.61   416.3 1012.13   447.5 1002.66
     455 1000.18   462.5 1001.68   513.1 1016.71   532.4 1023.62   551.8 1027.42
   609.9 1049.32   658.3 1062.27   677.7 1069.63     697 1072.76   735.7 1086.65
   784.1 1096.46   822.9 1109.57   842.2 1111.99   890.6 1126.83     910 1130.19
#Mann= 3 , 0 , 0
       0      .1       0   447.5    .045       0   462.5      .1       0
#XS Ineff= 2 , 0
          406.55 1013.63
Permanent Ineff=
       F       F
Bank Sta=447.5,462.5
XS Rating Curve= 0 ,0
Exp/Cntr=0.3,0.1

Type RM Length L Ch R = 1 ,8431.7  ,397.397,400,403.008
XS GIS Cut Line= 3
     1717993.845      380554.192     1717624.697      380288.364
     1717254.036      380024.298
#Sta/Elev= 30
       0  1084.1      29 1074.38    58.1 1059.25   125.8 1029.43   154.9 1019.19
   183.9 1002.61   203.3  999.62     242  998.39   309.7  998.51   387.1 1011.59
   396.8 1012.05   425.9 1009.33   447.4 1003.52   454.9 1000.82   462.4 1003.95
   474.3 1010.84     484    1014     542 1041.52   561.4 1048.35   590.5 1065.22
   638.9 1085.82   658.2 1097.77   677.6 1104.39   716.3 1121.97   735.7 1132.49
   784.1  1150.6   803.5 1160.52   822.9 1166.94   842.2 1176.59     910 1205.62
#Mann= 3 , 0 , 0
       0      .1       0   447.4    .045       0   462.4      .1       0
#XS Ineff= 2 , 0
           403.9 1012.76
Permanent Ineff=
       F       F
Bank Sta=447.4,462.4
XS Rating Curve= 0 ,0
Exp/Cntr=0.3,0.1

Type RM Length L Ch R = 1 ,8031.7  ,399.843,400,399.711
XS GIS Cut Line= 3
     1718201.626       380276.12     1717865.327       379969.18
     1717533.329       379658.23
#Sta/Elev= 30
       0 1023.49   164.7 1004.41   203.4  994.35   213.1  994.02   261.6  998.43
   377.8 1012.49   387.5 1012.53   426.2 1008.24   447.8 1002.17   455.3 1000.58
   462.8 1001.35     465 1001.57   474.7  1007.9   484.3 1012.63   513.4 1025.01
   532.7 1029.93   561.8 1042.57   581.1  1048.2   639.2 1071.39   706.9 1094.56
     736 1109.01   745.7 1111.28   774.7 1123.75   784.4  1126.6   803.7 1134.91
   823.1 1141.51   852.1 1156.04   871.5 1161.51   890.8 1170.75   910.2 1177.56
#Mann= 3 , 0 , 0
       0      .1       0   447.8    .045       0   462.8      .1       0
#XS Ineff= 2 , 0
          379.98 1012.83
Permanent Ineff=
       F       F
Bank Sta=447.8,462.8
XS Rating Curve= 0 ,0
Exp/Cntr=0.3,0.1

Type RM Length L Ch R = 1 ,7631.7  ,399.171,400,401.031
XS GIS Cut Line= 3
     1718471.638       379985.69     1718137.694       379676.63
     1717801.622      379369.908
#Sta/Elev= 30
       0 1037.52    19.4 1030.01    38.7 1024.02    77.4 1017.67    96.8 1011.48
   135.5 1003.26   222.7  993.49   271.1  999.02   387.2 1009.73   406.6 1008.46
   447.5  999.79     455  999.36   462.5  1000.6   474.4  1006.4   484.1 1013.29
   513.1 1029.57   542.1 1051.73   551.8 1061.75   561.5 1069.27   571.2 1072.91
   600.2 1088.82     668 1105.13   687.4 1107.31   716.4 1114.53   735.8 1117.38
   784.2 1130.64   813.2 1135.75   832.6 1140.38   851.9 1143.19     910 1156.17
#Mann= 3 , 0 , 0
       0      .1       0   447.5    .045       0   462.5      .1       0
#XS Ineff= 2 , 0
           397.7 1010.32
Permanent Ineff=
       F       F
Bank Sta=447.5,462.5
XS Rating Curve= 0 ,0
Exp/Cntr=0.3,0.1

Type RM Length L Ch R = 1 ,7231.7  ,361.561,358.426,352.756
XS GIS Cut Line= 3
     1718738.904      379711.351     1718416.496      379390.129
     1718177.541      379151.087
#Sta/Elev= 30
       0 1083.02    19.4 1071.22    58.1  1052.9    77.5 1045.86    96.8 1036.83
   116.2 1030.68   145.2 1017.85   164.6 1012.49   203.3  997.06   232.4  992.63
   242.1  992.35   271.1  996.26     397 1007.83   447.6  996.83   455.1  995.91
   462.6  997.53   464.8     998   484.1 1014.39   503.4 1023.52   532.4 1043.79
   551.7 1049.61     571  1058.6   619.3 1075.48   638.6  1079.1   667.6  1081.9
   706.2  1078.3   715.9  1078.4   744.8 1074.45   773.8 1072.96   793.1 1070.33
#Mann= 3 , 0 , 0
       0      .1       0   447.6    .045       0   462.6      .1       0
#XS Ineff= 2 , 0
          397.52 1007.79
Permanent Ineff=
       F       F
Bank Sta=447.6,462.6
XS Rating Curve= 0 ,0
Exp/Cntr=0.3,0.1

Type RM Length L Ch R = 1 ,6873.3  ,647.064,656.997,669.418
XS GIS Cut Line= 3
     1719018.789      379396.589     1718639.324      379111.494
       1718270.5      379081.368
#Sta/Elev= 30
       0 1098.29     9.7 1095.38    58.1 1074.48    87.2 1065.06   106.5 1056.36
   125.9 1050.59   145.3 1042.73   164.7 1036.64     184 1025.49   193.7 1022.32
   203.4  1017.1   222.8 1005.28   232.5 1001.92   251.8  992.24   261.5  989.86
   271.2  989.41     339  995.16   368.1 1000.56   406.8 1005.06   416.5 1004.03
   448.4  995.99   463.4   995.7   513.6  1007.5   523.3 1008.82   542.8 1010.26
     611 1011.57   679.1  1015.5   708.3 1018.47   786.3 1030.57   844.7 1035.06
#Mann= 3 , 0 , 0
       0      .1       0   448.4    .045       0   463.4      .1       0
#XS Ineff= 2 , 0
          417.18 1004.16
Permanent Ineff=
       F       F
Bank Sta=448.4,463.4
XS Rating Curve= 0 ,0
Exp/Cntr=0.3,0.1

Type RM Length L Ch R = 1 ,6216.3  ,184.147,184.577,183.973
XS GIS Cut Line= 3
      1719409.25      379337.006     1719231.079      378918.689
     1718961.419      378408.132
#Sta/Elev= 30
       0 1158.88      29 1154.64    67.7 1144.79    96.7 1134.82   203.2 1105.36
   232.2 1093.97   241.9 1093.01   309.6 1067.51   328.9 1062.66   348.3 1054.33
   377.3 1045.48   396.6 1037.01     416 1031.26   435.3  1021.6   454.7 1016.31
   474.3 1007.24   513.4  995.07   541.1   990.1   552.5   989.5   556.1  990.14
     621 1003.49   689.6  993.25   718.9  992.47     807  995.02   865.7 1016.42
   914.6 1036.89   934.2 1042.53   963.6 1058.92   983.1 1065.51  1032.1 1088.85
#Mann= 3 , 0 , 0
       0      .1       0   541.1    .045       0   556.1      .1       0
#XS Ineff= 2 , 0
                          626.04         1003.68
Permanent Ineff=
       F       F
Bank Sta=541.1,556.1
XS Rating Curve= 0 ,0
Exp/Cntr=0.3,0.1

Type RM Length L Ch R = 1 ,6031.7  ,454.521,449.759,446.03
XS GIS Cut Line= 3
     1719542.858      379140.021      1719339.65      378732.494
      1719117.84      378334.429
#Sta/Elev= 30
       0 1098.12    38.8 1099.06    67.8 1098.45    77.5 1096.83   106.6 1087.16
     126 1083.16   145.3 1075.64   164.7  1071.2   193.8 1060.63   203.5 1059.64
   251.9 1045.93   271.3 1038.12     281  1036.6   339.1 1018.37   358.5 1011.04
   377.9 1007.29   406.9  997.67   447.9  989.46   455.4  988.97   462.9  989.07
   542.6 1002.71   552.3 1002.01   581.4  994.06   620.2  991.76     659  991.05
   736.6  994.81   775.3 1004.92   804.4 1017.92   823.8 1022.65   911.1 1059.79
#Mann= 3 , 0 , 0
       0      .1       0   447.9    .045       0   462.9      .1       0
#XS Ineff= 2 , 0
                           552.7         1001.63
Permanent Ineff=
       F       F
Bank Sta=447.9,462.9
XS Rating Curve= 0 ,0
Exp/Cntr=0.3,0.1

Type RM Length L Ch R = 1 ,5582    ,353.588,350.241,346.682
XS GIS Cut Line= 3
      1719890.53       378861.71     1719757.847      378546.852
     1719399.632      378093.914
#Sta/Elev= 30
       0 1043.97     9.8 1043.42   117.1 1024.04   146.4 1023.52     166 1021.78
   214.8 1008.34   263.6  999.76   292.9  998.41   341.7 1000.36     371  998.86
     420     990   451.9  988.32   466.9  988.46   478.7  991.07   498.3   998.1
   517.9 1001.49   537.4  999.58     557   992.5   586.4  988.87   733.2  987.42
     743  987.58   762.5   990.7   772.3   993.5   791.9 1004.01   801.7 1007.23
   821.3 1010.05   870.2 1020.86   899.6 1030.81   909.4 1031.94   919.1 1035.45
#Mann= 3 , 0 , 0
       0      .1       0   451.9    .045       0   466.9      .1       0
#XS Ineff= 2 , 0
                          538.53          999.62
Permanent Ineff=
       F       F
Bank Sta=451.9,466.9
XS Rating Curve= 0 ,0
Exp/Cntr=0.3,0.1

Type RM Length L Ch R = 1 ,5231.7  ,398.849,400,401.364
XS GIS Cut Line= 3
     1720293.481      378550.237     1719960.891       378240.76
     1719622.798      377932.068
#Sta/Elev= 30
       0  1132.2      29 1121.88      58 1113.68    77.3 1105.97    96.7 1102.84
   193.3 1072.27   212.7 1068.49   251.3 1054.97   280.3 1048.24     319 1035.62
   328.6 1032.17   357.6 1012.33   367.3 1007.36     406 1004.41     435  995.08
   446.8  989.49   454.3  986.79   461.8  986.95   473.8  988.38     503  995.42
   532.2  999.53   580.9  991.13   590.7  990.59   795.2   986.4     805   987.2
   834.2   999.5   853.7 1003.44   873.2 1012.23   902.4 1021.66   912.1  1026.1
#Mann= 3 , 0 , 0
       0      .1       0   446.8    .045       0   461.8      .1       0
#XS Ineff= 2 , 0
                          535.87          999.58
Permanent Ineff=
       F       F
Bank Sta=446.8,461.8
XS Rating Curve= 0 ,0
Exp/Cntr=0.3,0.1

Type RM Length L Ch R = 1 ,4831.7  ,388.87,400,411.182
XS GIS Cut Line= 3
     1720558.973      378284.346     1720242.197       377957.73
     1719925.421      377631.114
#Sta/Elev= 30
       0 1030.86    48.4 1023.91    67.8 1022.25   135.5 1011.49   164.6 1009.01
   183.9 1008.69   222.7 1012.32   261.4 1013.96   300.1 1011.98   338.8    1006
   358.2 1001.83   406.6  996.87   447.5   986.1     455  985.06   462.5  985.59
   493.7  991.08   513.1   996.2   522.8  997.03   542.1  994.47   561.5  987.96
   571.2  986.32   600.2  987.33   716.4  986.54   726.1  988.34   735.7  991.98
   755.1  995.89   784.1 1006.76   813.2 1014.57   842.2 1024.69     910 1044.83
#Mann= 3 , 0 , 0
       0      .1       0   447.5    .045       0   462.5      .1       0
#XS Ineff= 2 , 0
                          522.59          997.13
Permanent Ineff=
       F       F
Bank Sta=447.5,462.5
XS Rating Curve= 0 ,0
Exp/Cntr=0.3,0.1

Type RM Length L Ch R = 1 ,4431.7  ,398.44,400,402.23
XS GIS Cut Line= 3
     1720710.375      378206.621     1720586.156      377768.906
     1720462.967      377330.899
#Sta/Elev= 30
       0 1071.62     9.7 1070.65    77.4 1056.13   135.5 1047.56   251.7 1026.99
   329.1 1007.28   358.2  995.12   396.9  993.69   416.3  990.22   435.6  983.43
   447.5  981.73     455  981.18   462.5  981.75   493.7  987.23   522.8  994.32
   532.4  995.07   542.1  994.17   561.5   987.9   580.9  986.23     697  986.02
   726.1  988.09   735.7  990.02   764.8 1001.14   774.5  1002.6   793.8 1010.09
   813.2 1014.67   842.2 1025.85   861.6 1031.11   900.3  1046.7     910 1052.82
#Mann= 3 , 0 , 0
       0      .1       0   447.5    .045       0   462.5      .1       0
#XS Ineff= 2 , 0
                          534.99          995.13
Permanent Ineff=
       F       F
Bank Sta=447.5,462.5
XS Rating Curve= 0 ,0
Exp/Cntr=0.3,0.1

Type RM Length L Ch R = 1 ,4031.7  ,398.201,400,403.33
XS GIS Cut Line= 3
     1721058.547      378095.104      1720964.86      377649.563
      1720885.59      377201.572
#Sta/Elev= 30
       0 1134.22    19.4 1128.94    38.7 1121.01    96.9 1106.26   125.9  1095.3
   164.7 1082.93   174.4 1081.43   203.4 1068.73   251.9 1054.98   280.9 1039.84
   300.3    1033   358.4  996.29   447.8  982.83   455.3  981.43   462.8  982.68
   484.3  990.57   503.7  993.56     523  992.03   552.1  986.22   648.9  984.79
   726.3  987.48     736  989.79   755.4 1000.09     765 1001.26   794.1 1015.95
   813.4 1022.24   832.8 1032.31   852.2 1038.05   871.5 1048.06   910.2 1063.17
#Mann= 3 , 0 , 0
       0      .1       0   447.8    .045       0   462.8      .1       0
#XS Ineff= 2 , 0
                          506.64          993.89
Permanent Ineff=
       F       F
Bank Sta=447.8,462.8
XS Rating Curve= 0 ,0
Exp/Cntr=0.3,0.1

Type RM Length L Ch R = 1 ,3631.7  ,408.661,400,388.739
XS GIS Cut Line= 3
     1721409.247      378005.244     1721351.312      377551.923
     1721338.932      377097.446
#Sta/Elev= 30
       0 1149.65    29.2 1137.23    87.5 1118.61   145.9 1095.54   165.3 1089.89
   194.5 1075.51   233.4 1060.69   243.1 1058.92     282 1042.07   311.2  1015.6
   320.9 1013.68   340.3  997.87     350  994.83   449.5  980.32     457  979.66
   464.5  981.94   505.4  992.54   553.7  986.03   582.8  985.89   602.1  988.64
   679.5  1014.9   698.8 1024.65   718.2 1030.08   756.9 1045.95   776.2 1056.21
   834.3 1076.75   863.3 1091.16     873 1092.09   892.3 1101.98   911.7 1107.82
#Mann= 3 , 0 , 0
       0      .1       0   449.5    .045       0   464.5      .1       0
#XS Ineff= 2 , 0
                          512.84          992.63
Permanent Ineff=
       F       F
Bank Sta=449.5,464.5
XS Rating Curve= 0 ,0
Exp/Cntr=0.3,0.1

Type RM Length L Ch R = 1 ,3231.7  ,406.515,400,396.206
XS GIS Cut Line= 3
     1721952.487       377842.83     1721729.979      377446.241
     1721500.544      377051.647
#Sta/Elev= 30
       0 1037.38    19.4 1037.59      29 1036.01    58.1 1029.51    77.4 1027.77
   116.1 1016.08   203.2 1005.62   261.2  994.01   280.6   992.1   406.4  988.12
   435.4  979.79   447.2  977.91   454.7  977.54   462.2  977.81   542.1  989.76
   551.9  989.31   571.3   984.3   590.7  981.55   600.4  981.74   619.8  991.01
   629.6  993.28   678.1 1011.08   707.2 1024.04   726.7 1030.31   755.8 1043.79
   775.2 1048.91   794.7 1058.96   814.1 1065.28   891.8 1098.22   911.2 1104.85
#Mann= 3 , 0 , 0
       0      .1       0   447.2    .045       0   462.2      .1       0
#XS Ineff= 2 , 0
                          548.27          989.89
Permanent Ineff=
       F       F
Bank Sta=447.2,462.2
XS Rating Curve= 0 ,0
Exp/Cntr=0.3,0.1

Type RM Length L Ch R = 1 ,2831.7  ,393.048,400,404.447
XS GIS Cut Line= 3
     1722338.317      377493.974     1722010.496       377174.28
      1721717.59      376823.317
#Sta/Elev= 30
       0 1145.14    29.2 1132.25    58.5 1122.21    87.7 1114.86   185.1 1080.88
   292.3 1034.85     302 1032.81   311.8 1027.64   331.2 1013.18   350.7 1004.65
   370.2  990.41     380  986.26   450.4  976.17   457.9  975.87   465.4  975.91
   545.4  988.89   584.3  980.54   594.1  981.18   652.4 1004.87   671.9 1010.03
   701.1 1023.84   720.5 1028.56   749.7 1041.81   769.1  1046.6   798.3 1060.73
   817.8 1066.77   846.9 1081.28   866.4 1086.93   905.3 1105.74     915 1108.57
#Mann= 3 , 0 , 0
       0      .1       0   450.4    .045       0   465.4      .1       0
#XS Ineff= 2 , 0
                          547.39          988.95
Permanent Ineff=
       F       F
Bank Sta=450.4,465.4
XS Rating Curve= 0 ,0
Exp/Cntr=0.3,0.1

Type RM Length L Ch R = 1 ,2431.7  ,399.473,400,400.658
XS GIS Cut Line= 3
     1722529.204      377327.913     1722313.994      376927.287
     1722095.734      376526.579
#Sta/Elev= 30
       0 1176.01    38.7  1158.3    48.4 1156.04    77.4 1140.92    96.8 1135.24
   125.8 1118.49   183.8 1095.74   212.9 1081.18   232.2 1075.69   270.9  1057.8
     300 1041.75   319.3 1034.21   338.7    1021   367.7 1007.85   396.7  989.88
   447.3  976.45   454.8  975.97   462.3  976.16   542.1  989.81   629.5 1015.75
   678.1 1032.65   697.5 1042.74   765.4 1069.14   784.9 1079.68   804.3 1085.55
   833.4 1099.58   843.1 1101.85   872.2 1117.05   891.6 1123.05   911.1 1132.67
#Mann= 3 , 0 , 0
       0      .1       0   447.3    .045       0   462.3      .1       0
Bank Sta=447.3,462.3
XS Rating Curve= 0 ,0
Exp/Cntr=0.3,0.1

Type RM Length L Ch R = 1 ,2031.7  ,401.774,400,397.993
XS GIS Cut Line= 3
     1722867.728      377137.399     1722661.891       376731.62
     1722456.054      376325.842
#Sta/Elev= 30
       0 1083.69    19.4 1084.03    38.7 1079.22   125.9 1069.24   193.6 1064.39
   222.7 1056.32   232.3 1055.63   290.4 1037.33   309.8 1025.05   319.5 1023.18
   348.5  999.31   358.2  994.75   387.2  987.24   447.5  975.95     455  975.76
   462.5  975.87   513.1  984.04   551.8  984.08   561.5   986.7   590.5  998.07
   609.9 1009.46   619.6 1012.59   648.6 1030.04   677.7 1041.88     697 1053.79
   706.7 1056.02   784.1 1089.67   803.5  1093.3     881 1119.21     910 1132.43
#Mann= 3 , 0 , 0
       0      .1       0   447.5    .045       0   462.5      .1       0
Bank Sta=447.5,462.5
XS Rating Curve= 0 ,0
Exp/Cntr=0.3,0.1
